--- D140-00-00.prj (project) ---

Proj Title=D140-00-00
Current Plan=p06
Default Exp/Contr=.3,.1
English Units
Geom File=g02
Flow File=f05
Flow File=f06
Flow File=f03
Plan File=p06
Plan File=p08
Plan File=p04
Y Axis Title=Elevation (
X Axis Title(PF)=STATION
X Axis Title(XS)=Station
BEGIN DESCRIPTION:
Brays Bayou Watershed
Fondren Diversion Channel
HCFCD Unit D140-00-00
Flood Hazard & Floodway Model
10, 2, 1, 0.2% Event
Filename D140.prj
Prepared by: Dodson & Associates, Inc.   Date: September 2003
Reviewed by:____________________	 Date:_________
STATUS (Final RAS, SVSQ
FOR FLOOD HARZARD RECOVERY DATA ONLY,03/02/2004
Will Be Voided Upon Release of The Preliminary DFIRM
END DESCRIPTION:
DSS Export Rating Curves= 0
DSS Export Rating Curve Sorted= 0
DSS Export Volume Flow Curves= 0
DXF OffsetX= 0
DXF OffsetY= 0
DXF ScaleX= 1
DXF ScaleY= 10

--- D140-00-00.p06 (plan) ---

Plan Title=FEMA Effective June 2007
Version=Version 3.0.1  Mar 2001
Short Identifier=FEMAeff0607
Geom File=g02
Flow File=f05
Subcritical Flow
K Sum by GR= 0
Std Step Tol= 0.01
Critical Tol= 0.01
Num of Std Step Trials= 20
Max Error Tol= 0.3
Flow Tol Ratio= 0.001
Split Flow NTrial= 30
Split Flow Tol= 0.02
Split Flow Ratio= 0.02
Log Output Level= 0
Friction Slope Method= 2
Unsteady Friction Slope Method= 2
Secant Critical Depth
Global Vel Dist= 0 , 0 , 0
Global Log Level= 0
CheckData=True
Encroach Param=-1 ,0,0, 0
Computation Interval=1HOUR
Output Interval=1HOUR
Run HTab= 0
Run UNet= 0
Run PostProcess= 0
UNET Theta= 1
UNET ZTol= 0.02
UNET ZSATol= 0.1
UNET MxIter= 20
UNET MaxInSteps= 20
UNET DtIC= 0
UNET DtMin= 0
UNET MaxCRTS= 20
UNET WFStab= 2
UNET SFStab= 1
UNET WFX= 1
UNET SFX= 1
UNET Convert EG Bridges=-1
UNET Use Existing IB Tables=-1
Instantaneous Interval=1HOUR
Write IC File= 0
Write Velocity= 0
Write Detailed= 0

--- D140-00-00.p04 (plan) ---

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Plan Title=Storage Routing
Short Identifier=Store_Rout
Geom File=g02
Flow File=f03

--- D140-00-00.p08 (plan) ---

Plan Title=Floodway
Version=Version 3.0.1  Mar 2001
Short Identifier=Floodway0607
Geom File=g02
Flow File=f06
Subcritical Flow
K Sum by GR= 0
Std Step Tol= 0.01
Critical Tol= 0.01
Num of Std Step Trials= 20
Max Error Tol= 0.3
Flow Tol Ratio= 0.001
Split Flow NTrial= 30
Split Flow Tol= 0.02
Split Flow Ratio= 0.02
Log Output Level= 0
Friction Slope Method= 2
Unsteady Friction Slope Method= 2
Secant Critical Depth
Global Vel Dist= 0 , 0 , 0
Global Log Level= 0
CheckData=True
Encroach Param=-1 ,0,0, 2
Encroach River=D140-00-00
Encroach Reach=Reach 0
Encroach Node=19911
       1 3629.14  3758.8
Encroach Node=18719
       1 4031.36 4135.94
Encroach Node=18310
       1 4138.32 4209.87
Encroach Node=17910
       1 4341.88 4409.39
Encroach Node=17874
       1 4343.88 4411.39
Encroach Node=17837
       1 4343.88 4450.25
Encroach Node=17793
       1 4381.88 4450.25
Encroach Node=17764
       1 4394.88 4462.39
Encroach Node=17698
       1 4442.82 4509.21
Encroach Node=17069
       1 4525.43 4594.99
Encroach Node=17034
       1 4574.43  4642.4
Encroach Node=17013
       1 4571.43  4642.4
Encroach Node=16996
       1 4571.43  4639.4
Encroach Node=16957
       1 4569.43 4639.43
Encroach Node=16707
       1 4628.43  4696.4
Encroach Node=16495
       1 4580.93 4726.34
Encroach Node=16480
       1 4536.82 4726.34
Encroach Node=16472
       1 4536.82  4689.3
Encroach Node=16368
       1 4451.25 4586.27
Encroach Node=16152
       1 4317.17 4466.49
Encroach Node=15749
       1 3968.58 4121.17
Encroach Node=15538
       1 3779.65 3947.33
Encroach Node=14872
       1 4215.48  4380.9
Encroach Node=14119
       1 4813.05 4976.46
Encroach Node=13655
       1 5285.76 5449.67
Encroach Node=13551
       1 5409.74 5615.16
Encroach Node=13459
       1 5482.23 5657.56
Encroach Node=13400
       1 5482.23 5766.56
Encroach Node=13347
       1 5605.22 5766.56
Encroach Node=13248
       1  5683.1 5898.92
Encroach Node=13169
       1 5751.04 5935.14
Encroach Node=12531
       1 6098.54 6239.68
Encroach Node=11781
       1 5850.75 6018.97
Encroach Node=11700
       1 5861.75 6024.35
Encroach Node=11650
       1 5810.64 6024.35
Encroach Node=11586
       1 5810.64 5952.35
Encroach Node=11502
       1 5771.64 5913.35
Encroach Node=10912
       1 5567.36 5710.96
Encroach Node=9302
       1 5319.12 5488.38
Encroach Node=9187
       1 5807.81 5979.38
Encroach Node=9164
       1 5807.81 6243.38
Encroach Node=9145
       1 6074.12 6243.38
Encroach Node=9025
       1 6057.43 6238.38
Encroach Node=8552
       1 6052.59 6218.37
Encroach Node=7849
       1 6007.11 6192.22
Encroach Node=7530
       1 5997.34  6180.9
Encroach Node=7427
       1 6040.78 6187.44
Encroach Node=7378
       1 6040.78 6187.44
Encroach Node=7329
       1 6041.78  6179.9
Encroach Node=7221
       1 6038.78  6176.9
Encroach Node=6446
       1 5999.84 6151.15
Encroach Node=5555
       1 5599.83 5799.32
Encroach Node=5032
       1 5431.82 5656.71
Encroach Node=4873
       1 5421.52 5637.99
Encroach Node=4862
       1 5419.17 5646.61
Encroach Node=4853
       1 5419.17 5646.61
Encroach Node=4694
       1 5396.86 5621.91
Encroach Node=4636
       1 5398.76  5623.8
Encroach Node=3724
       1 5123.98 5354.92
Encroach Node=3589
       1 3969.82 4147.26
Encroach Node=3546
       1  3743.6 4147.26
Encroach Node=3504
       1  3743.6 3920.26
Encroach Node=3392
       1  193.01  475.86
Encroach Node=3104
       1  263.09  435.69
Encroach Node=2212
       1  257.75  458.35
Encroach Node=2137
       1  191.12  454.48
Encroach Node=2011
       1  266.29  428.58
Encroach Node=1970
       1  266.29  428.58
Encroach Node=1931
       1  266.29  428.58
Encroach Node=1802
       1  261.29  423.58
Encroach Node=1374
       1  248.67  421.73
Encroach Node=837
       1  242.94  457.37
Encroach Node=370
       1  234.48  445.74
Encroach Node=295
       1  234.48  445.74
Encroach Node=268
       1  238.06  436.64
Encroach Node=178
       1  238.06  436.64
Encroach Node=122
       1  168.29  361.89
Encroach Node=102
       1  168.29  361.89
Encroach Reach=D140-00-00_0001
Encroach Node=19911
       1 3629.14  3758.8
Encroach Node=18719
       1 4031.36 4135.94
Encroach Node=18310
       1 4138.32 4209.87
Encroach Node=17910
       1 4341.88 4409.39
Encroach Node=17874
       1 4343.88 4411.39
Encroach Node=17837
       1 4343.88 4450.25
Encroach Node=17793
       1 4381.88 4450.25
Encroach Node=17764
       1 4394.88 4462.39
Encroach Node=17698
       1 4442.82 4509.21
Encroach Node=17069
       1 4525.43 4594.99
Encroach Node=17034
       1 4574.43  4642.4
Encroach Node=17013
       1 4571.43  4642.4
Encroach Node=16996
       1 4571.43  4639.4
Encroach Node=16957
       1 4569.43 4639.43
Encroach Node=16707
       1 4628.43  4696.4
Encroach Node=16495
       1 4580.93 4726.34
Encroach Node=16480
       1 4536.82 4726.34
Encroach Node=16472
       1 4536.82  4689.3
Encroach Node=16368
       1 4451.25 4586.27
Encroach Node=16152
       1 4317.17 4466.49
Encroach Node=15749
       1 3968.58 4121.17
Encroach Node=15538
       1 3779.65 3947.33
Encroach Node=14872
       1 4215.48  4380.9
Encroach Node=14119
       1 4813.05 4976.46
Encroach Node=13655
       1 5285.76 5449.67
Encroach Node=13551
       1 5409.74 5615.16
Encroach Node=13459
       1 5482.23 5657.56
Encroach Node=13400
       1 5482.23 5766.56
Encroach Node=13347
       1 5605.22 5766.56
Encroach Node=13248
       1  5683.1 5898.92
Encroach Node=13169
       1 5751.04 5935.14
Encroach Node=12531
       1 6098.54 6239.68
Encroach Node=11781
       1 5850.75 6018.97
Encroach Node=11700
       1 5861.75 6024.35
Encroach Node=11650
       1 5810.64 6024.35
Encroach Node=11586
       1 5810.64 5952.35
Encroach Node=11502
       1 5771.64 5913.35
Encroach Node=10912
       1 5567.36 5710.96
Encroach Node=9302
       1 5319.12 5488.38
Encroach Node=9187
       1 5807.81 5979.38
Encroach Node=9164
       1 5807.81 6243.38
Encroach Node=9145
       1 6074.12 6243.38
Encroach Node=9025
       1 6057.43 6238.38
Encroach Node=8552
       1 6052.59 6218.37
Encroach Node=7849
       1 6007.11 6192.22
Encroach Node=7530
       1 5997.34  6180.9
Encroach Node=7427
       1 6040.78 6187.44
Encroach Node=7378
       1 6040.78 6187.44
Encroach Node=7329
       1 6041.78  6179.9
Encroach Node=7221
       1 6038.78  6176.9
Encroach Node=6446
       1 5999.84 6151.15
Encroach Node=5555
       1 5599.83 5799.32
Encroach Node=5032
       1 5431.82 5656.71
Encroach Node=4873
       1 5421.52 5637.99
Encroach Node=4862
       1 5419.17 5646.61
Encroach Node=4853
       1 5419.17 5646.61
Encroach Node=4694
       1 5396.86 5621.91
Encroach Node=4636
       1 5398.76  5623.8
Encroach Node=3724
       1 5123.98 5354.92
Encroach Node=3589
       1 3969.82 4147.26
Encroach Node=3546
       1  3743.6 4147.26
Encroach Node=3504
       1  3743.6 3920.26
Encroach Node=3392
       1  193.01  475.86
Encroach Node=3104
       1  263.09  435.69
Encroach Node=2212
       1  257.75  458.35
Encroach Node=2137
       1  191.12  454.48
Encroach Node=2011
       1  266.29  428.58
Encroach Node=1970
       1  266.29  428.58
Encroach Node=1931
       1  266.29  428.58
Encroach Node=1802
       1  261.29  423.58
Encroach Node=1374
       1  248.67  421.73
Encroach Node=837
       1  242.94  457.37
Encroach Node=370
       1  234.48  445.74
Encroach Node=295
       1  234.48  445.74
Encroach Node=268
       1  238.06  436.64
Encroach Node=178
       1  238.06  436.64
Encroach Node=122
       1  168.29  361.89
Encroach Node=102
       1  168.29  361.89
Computation Interval=1HOUR
Output Interval=1HOUR
Run HTab= 0
Run UNet= 0
Run PostProcess= 0
UNET Theta= 1
UNET ZTol= 0.02
UNET ZSATol= 0.1
UNET MxIter= 20
UNET MaxInSteps= 20
UNET DtIC= 0
UNET DtMin= 0
UNET MaxCRTS= 20
UNET WFStab= 2
UNET SFStab= 1
UNET WFX= 1
UNET SFX= 1
UNET Convert EG Bridges=-1
UNET Use Existing IB Tables=-1
Instantaneous Interval=1HOUR
Write IC File= 0
Write Velocity= 0
Write Detailed= 0

--- D140-00-00.f05 (steady flow) ---

Flow Title=FEMA Effective June 2007
Version=Version 3.0.1  Mar 2001
Number of Profiles= 4
Profile Names=10PCT_10yr,2PCT_50yr,1PCT_100yr,0.2PCT_500yr
River Rch & RM=D140-00-00,D140-00-00_0001 ,19911
    1491    2235    2609    3669
River Rch & RM=D140-00-00,D140-00-00_0001 ,18719
    1573    2359    2751    3846
River Rch & RM=D140-00-00,D140-00-00_0001 ,17698
    1634    2453    2858    3980
River Rch & RM=D140-00-00,D140-00-00_0001 ,16957
    1777    2671    3108    4290
River Rch & RM=D140-00-00,D140-00-00_0001 ,15538
    1893    2848    3310    4539
River Rch & RM=D140-00-00,D140-00-00_0001 ,14119
    1989    2995    3477    4743
River Rch & RM=D140-00-00,D140-00-00_0001 ,13169
    2236    3373    3908    5265
River Rch & RM=D140-00-00,D140-00-00_0001 ,10912
    2574    3870    4356    5555
River Rch & RM=D140-00-00,D140-00-00_0001 ,9025
    2809    4216    4661    5744
River Rch & RM=D140-00-00,D140-00-00_0001 ,7849
    2944    4413    4832    5848
River Rch & RM=D140-00-00,D140-00-00_0001 ,7221
    3072    3885    4183    5033
River Rch & RM=D140-00-00,D140-00-00_0001 ,5555
    3152    4009    4331    5228
River Rch & RM=D140-00-00,D140-00-00_0001 ,4636
    3291    4224    4590    5569
River Rch & RM=D140-00-00,D140-00-00_0001 ,3104
    3456    4480    4901    5980
River Rch & RM=D140-00-00,D140-00-00_0001 ,1374
    3592    4695    5163    6329
Boundary for River Rch & Prof#=D140-00-00,D140-00-00_0001 , 1
Up Type= 0
Dn Type= 3
Dn Slope=.0006
Boundary for River Rch & Prof#=D140-00-00,D140-00-00_0001 , 2
Up Type= 0
Dn Type= 3
Dn Slope=.0006
Boundary for River Rch & Prof#=D140-00-00,D140-00-00_0001 , 3
Up Type= 0
Dn Type= 3
Dn Slope=.0006
Boundary for River Rch & Prof#=D140-00-00,D140-00-00_0001 , 4
Up Type= 0
Dn Type= 3
Dn Slope=.0006
DSS Import GetInterval= 0
DSS Import GetPeak= 0
DSS Import FillOption= 0

--- D140-00-00.f03 (steady flow) ---

Flow Title=Storage Routing
Version=Version 3.0.1  Mar 2001
Number of Profiles= 8
Profile Names=0.1,0.2,0.4,0.6,0.8,1.0,1.2,1.5
River Rch & RM=D140-00-00,D140-00-00_0001 ,19911
     391     782    1564    2346    3128    3910    4692    5865
River Rch & RM=D140-00-00,D140-00-00_0001 ,10912
     432     864    1728    2592    3456    4320    5184    6480
River Rch & RM=D140-00-00,D140-00-00_0001 ,7221
     517    1034    2068    3102    4136    5170    6204    7755
Boundary for River Rch & Prof#=D140-00-00,D140-00-00_0001 , 1
Up Type= 0
Dn Type= 3
Dn Slope=.0006
Boundary for River Rch & Prof#=D140-00-00,D140-00-00_0001 , 2
Up Type= 0
Dn Type= 3
Dn Slope=.0006
Boundary for River Rch & Prof#=D140-00-00,D140-00-00_0001 , 3
Up Type= 0
Dn Type= 3
Dn Slope=.0006
Boundary for River Rch & Prof#=D140-00-00,D140-00-00_0001 , 4
Up Type= 0
Dn Type= 3
Dn Slope=.0006
Boundary for River Rch & Prof#=D140-00-00,D140-00-00_0001 , 5
Up Type= 0
Dn Type= 3
Dn Slope=.0006
Boundary for River Rch & Prof#=D140-00-00,D140-00-00_0001 , 6
Up Type= 0
Dn Type= 3
Dn Slope=.0006
Boundary for River Rch & Prof#=D140-00-00,D140-00-00_0001 , 7
Up Type= 0
Dn Type= 3
Dn Slope=.0006
Boundary for River Rch & Prof#=D140-00-00,D140-00-00_0001 , 8
Up Type= 0
Dn Type= 3
Dn Slope=.0006
DSS Import GetInterval= 0
DSS Import GetPeak= 0
DSS Import FillOption= 0

--- D140-00-00.f06 (steady flow) ---

Flow Title=Floodway
Version=Version 3.0.1  Mar 2001
Number of Profiles= 2
Profile Names=1PCT_100yr,1PCTFloodway_100yrFW
River Rch & RM=D140-00-00,D140-00-00_0001 ,19911
    2609    2609
River Rch & RM=D140-00-00,D140-00-00_0001 ,18719
    2751    2751
River Rch & RM=D140-00-00,D140-00-00_0001 ,17698
    2858    2858
River Rch & RM=D140-00-00,D140-00-00_0001 ,16957
    3108    3108
River Rch & RM=D140-00-00,D140-00-00_0001 ,15538
    3310    3310
River Rch & RM=D140-00-00,D140-00-00_0001 ,14119
    3477    3477
River Rch & RM=D140-00-00,D140-00-00_0001 ,13169
    3908    3908
River Rch & RM=D140-00-00,D140-00-00_0001 ,10912
    4356    4356
River Rch & RM=D140-00-00,D140-00-00_0001 ,9025
    4661    4661
River Rch & RM=D140-00-00,D140-00-00_0001 ,7849
    4832    4832
River Rch & RM=D140-00-00,D140-00-00_0001 ,7221
    4183    4183
River Rch & RM=D140-00-00,D140-00-00_0001 ,5555
    4331    4331
River Rch & RM=D140-00-00,D140-00-00_0001 ,4636
    4590    4590
River Rch & RM=D140-00-00,D140-00-00_0001 ,3104
    4901    4901
River Rch & RM=D140-00-00,D140-00-00_0001 ,1374
    5163    5163
Boundary for River Rch & Prof#=D140-00-00,D140-00-00_0001 , 1
Up Type= 0
Dn Type= 1
Dn Known WS=53.88
Boundary for River Rch & Prof#=D140-00-00,D140-00-00_0001 , 2
Up Type= 0
Dn Type= 1
Dn Known WS=53.88
DSS Import GetInterval= 0
DSS Import GetPeak= 0
DSS Import FillOption= 0

--- D140-00-00.g02 (geometry) ---

Geom Title=D140-00-00 June 2007
Version=Version 3.0.1  Mar 2001

River Reach=D140-00-00      ,D140-00-00_0001
Reach XY= 30
      3071706.52    13796722.829     3071894.972    13796723.129
     3071949.281    13795918.584       3072232.5    13795932.093
     3075262.379    13796076.601     3075367.331    13796191.948
     3075384.486    13796941.507     3075419.167    13797263.673
     3075428.661    13797328.238     3075452.922    13797355.119
       3077287.5    13797449.718     3077294.597    13797450.083
       3078202.5    13797484.273     3078216.096    13797484.784
     3078329.883    13797516.282     3078377.086    13797595.607
      3078339.52    13798324.134     3078285.743    13799615.691
     3078219.801      13801282.5     3078214.006    13801429.006
      3078210.58     13801515.58     3078201.249    13801751.467
     3078200.059      13801777.5     3078198.201    13801818.201
     3078194.269    13801904.269     3078187.063    13802062.063
     3078183.131    13802148.131     3078101.979    13803924.927
     3078028.667    13806366.104     3077851.864    13810027.468

Type RM Length L Ch R = 1 ,19911   ,1179.38,1192.44,1207.88
BEGIN DESCRIPTION:
19911.20  Survey
END DESCRIPTION:
XS GIS Cut Line= 5
      3071459.42    13799551.187     3072044.084     13797488.65
     3072105.859    13796004.593     3072105.859    13795874.934
     3072157.377    13794130.367
#Sta/Elev= 30
       0   66.81  118.17   66.51  149.35   64.35  211.71   66.94  304.63   66.62
  390.15   63.97  461.17   66.75  570.31    66.7  617.08   63.48  705.99   66.64
  866.54   64.13 1006.85   66.55 1129.65   63.49 1225.13    65.8 2030.07   65.61
  2139.4   63.67 2250.04   65.87 2475.24   62.21  2550.3   64.55  2715.1   61.05
 3361.01   61.59 3629.14   64.05 3703.32   49.12 3709.17   49.23 3749.91   62.98
  3758.8   63.53 4603.32   65.16 4801.69   63.31 5084.33   66.02 5504.13   64.91
#Mann= 3 , 0 , 0
       0     .15       0 3629.14     .04       0  3758.8     .15       0
#XS Ineff= 2 , 0
       0    3618            3784       0
Permanent Ineff=
       T       T
Bank Sta=3629.14,3758.8
XS Rating Curve= 0
Exp/Cntr=.3,.1

Type RM Length L Ch R = 1 ,18719   ,413.99,408.38,400.34
BEGIN DESCRIPTION:
18718.76  Survey
END DESCRIPTION:
XS GIS Cut Line= 6
     3071692.704    13799542.854     3073241.209    13797518.439
     3073283.249    13796059.791     3073310.595    13795906.193
     3073441.919    13793597.123     3073480.507    13792919.374
#Sta/Elev= 30
       0   67.37  415.92    67.2  577.92   64.55 1070.14   67.24  1283.5   63.61
 1444.64   66.94 1643.45   63.33 1840.56   66.32 1983.38   62.84 2096.69   65.62
 2304.43   63.44 2542.65   66.05 2744.77   63.46 2849.82   65.65 2939.85   62.98
 3345.02   63.04 3450.06   66.07 3596.24   63.11 3765.19   65.33 3840.23   62.37
 4031.36   63.92 4086.03   46.35 4135.94   62.42 4563.36   66.46 5134.28   64.36
 5179.35   69.67  5209.4   64.14 5254.25   63.81 5936.82   66.65 7155.67   65.79
#Mann= 3 , 0 , 0
       0     .15       0 4031.36     .04       0 4135.94     .15       0
#XS Ineff= 2 , 0
       0    4008            4157       0
Permanent Ineff=
       T       T
Bank Sta=4031.36,4135.94
XS Rating Curve= 0
Exp/Cntr=.3,.1

Type RM Length L Ch R = 1 ,18310   ,409.78,400.82,381.5
BEGIN DESCRIPTION:
18310.38  Survey
END DESCRIPTION:
XS GIS Cut Line= 5
     3071965.001    13799569.912     3073632.948     13797549.09
      3073699.79    13796029.914     3073714.546    13795949.608
     3073737.974    13792683.728
#Sta/Elev= 30
       0   66.53  593.07   65.04  773.69   67.54  949.67   63.92 1115.16   67.31
 1328.26   64.14 1455.35   67.08 2077.74   63.51 2466.73   66.16 2832.06    62.3
 2932.96   65.44 4138.32   64.09 4178.52   50.69 4179.18   46.67 4186.45   46.67
 4187.11   50.68 4209.87   62.92 4977.23    64.6 5279.69   61.49 5349.56   64.36
 5819.71   62.57 5954.71   65.65 6089.71   62.51 6194.72   66.49 6344.72   62.98
 6449.72   66.42 6614.73   63.17 6659.73   66.51 7017.64    67.9 7488.52    66.1
#Mann= 3 , 0 , 0
       0     .15       0 4138.32    .017       0 4209.87     .15       0
#XS Ineff= 2 , 0
       0    4133            4210       0
Permanent Ineff=
       T       T
Bank Sta=4138.32,4209.87
XS Rating Curve= 0
Exp/Cntr=.3,.1

Type RM Length L Ch R = 1 ,17910   ,35.57,35.33,36.4
BEGIN DESCRIPTION:
 17909.56
END DESCRIPTION:
XS GIS Cut Line= 5
     3072064.177    13799580.929     3074020.709    13797568.578
     3074109.496    13796069.256      3074101.56     13795980.36
     3073942.836    13792496.228
#Sta/Elev= 30
       0   67.79 1015.97   64.33 1575.58   67.44  1726.2   63.52 2285.67   66.16
 2522.28   62.69 3203.47   65.28 3320.12   61.95 3788.26   65.15 4341.88   61.63
 4365.26   50.37 4366.19   46.32 4373.26   46.32 4374.19   50.39 4409.39   62.34
 5366.76   64.14 5482.17   61.27 5560.83   64.27 5922.34   65.47 6017.06   62.44
 6190.12   65.59 6282.71   61.93 6417.85   65.92 6522.96   61.83 6688.13   66.07
 6803.68   62.33 6882.34   66.21 7196.98   67.66 7779.08   62.65 7885.64   66.58
#Mann= 3 , 0 , 0
       0     .15       0 4341.88    .017       0 4409.39     .15       0
#XS Ineff= 2 , 0
       0    4318            4430       0
Permanent Ineff=
       T       T
Bank Sta=4341.88,4409.39
XS Rating Curve= 0
Exp/Cntr=.5,.3

Type RM Length L Ch R = 1 ,17874   ,81.49,81.6,80.44
BEGIN DESCRIPTION:
 17874.24
END DESCRIPTION:
XS GIS Cut Line= 5
     3072133.576    13799600.757     3074068.665    13797588.294
      3074144.44    13796067.096     3074136.504      13795978.2
     3074012.255    13792432.693
#Sta/Elev= 30
       0   68.86  640.48   64.69 1469.07   67.12 1606.98    63.2 1765.83   66.65
 1946.46   63.33 3253.24   64.96 3325.61   61.51 3433.46   64.68 3583.12   61.98
 3793.91   65.06 4343.88   61.63 4367.26   50.37 4368.19   46.32 4375.26   46.32
 4376.19   50.39 4411.39   62.34 5460.56   61.31 5919.92   64.19 6013.25   61.61
 6196.01   65.18 6271.06   61.48 6448.77   64.95 6541.22   61.61 6691.31   66.01
 6781.37   61.91 6930.95   66.18 7724.22   66.06 7801.99    62.1 7951.89   64.92
#Mann= 3 , 0 , 0
       0     .15       0 4343.88    .017       0 4411.39     .15       0
#XS Ineff= 2 , 0
       0    4320            4420       0
Permanent Ineff=
       T       T
Bank Sta=4343.88,4411.39
XS Rating Curve= 0
Exp/Cntr=.5,.3

Type RM Length L Ch R = 3 ,17837   ,,,
BEGIN DESCRIPTION:
McLain Bridge
END DESCRIPTION:
Bridge Culvert--1,0,-1,-1, 0
Deck Dist Width WeirC Skew NumUp NumDn MinLoCord MaxHiCord MaxSubmerge Is_Ogee
5,64,2.6,0, 8, 8, , , .95, 0, 0,0,,
    4330 4344.64 4352.33 4352.33 4374.83 4397.33 4397.33    4412
    62.1   62.45   62.37   62.37   62.36    62.3    62.3    62.3
       0       0       0   60.27   60.26    60.2       0       0
    4360 4382.64 4390.33 4390.33 4412.83 4435.33 4435.33    4450
   62.08   62.45   62.37   62.37   62.36    62.3    62.3    62.3
       0       0       0   60.27   60.26    60.2       0       0
BR Coef=-1 , 0 , 0 ,, 0 ,,,.8,-1,,0,
WSPro=,,,, 1 ,,,, 0 ,,,, 0 ,,,,-1 ,-1 ,-1 , 0 , 0 , 0 , 0 , 0
BC Design=,, 0 ,, 0 ,,,,,,

Type RM Length L Ch R = 1 ,17793   ,29.34,28.42,29.74
BEGIN DESCRIPTION:
17792.63  Survey
END DESCRIPTION:
XS GIS Cut Line= 5
     3072173.232    13799600.757     3074166.998    13797588.243
     3074225.156    13796062.106     3074217.221    13795973.209
     3074065.454    13792384.002
#Sta/Elev= 30
       0   67.21  335.38   65.26  440.95    67.6  673.21   64.87  863.25   67.17
 1000.68   63.76 1341.69   67.09 1448.26   64.05  1652.9   66.55 1831.89   63.14
 2193.47   66.15 2404.61   62.35 2565.08   65.07 2830.24    63.2 2944.96   65.09
 2993.76   62.66 3320.91   61.41 4381.88   61.63 4405.26   50.37 4406.19   46.32
 4413.26   46.32 4414.19   50.39 4450.25   62.33 6852.25   60.83 7152.51   64.99
 7251.25   63.38 7798.09   65.96 7873.16   61.96 7963.24   64.68  8041.8   63.17
#Mann= 3 , 0 , 0
       0     .15       0 4381.88    .017       0 4450.25     .15       0
#XS Ineff= 2 , 0
       0    4355            4455       0
Permanent Ineff=
       T       T
Bank Sta=4381.88,4450.25
XS Rating Curve= 0
Exp/Cntr=.5,.3

Type RM Length L Ch R = 1 ,17764   ,65.81,66.51,76.17
BEGIN DESCRIPTION:
 17764.22
END DESCRIPTION:
XS GIS Cut Line= 5
     3072222.802    13799610.671     3074214.444    13797627.832
     3074253.267    13796060.366     3074245.331     13795971.47
     3074142.884    13792313.134
#Sta/Elev= 30
       0   66.82  808.13   66.49  902.67   64.19 1539.99   66.47 1741.52   63.36
 2137.62   66.12 2299.65   62.87 2505.19    65.1 2780.97   62.28 2945.47   65.15
 3004.04   62.52 3160.83   64.65 3355.45   61.54  3443.3   63.79 4301.18   63.98
 4394.88   61.63 4418.26   50.37 4419.19   46.32 4426.26   46.32 4427.19   50.39
 4462.39   62.34 5636.92   64.16 5727.05   60.94 5930.24   65.46  6867.5   61.04
 7842.88   66.09 7962.93   61.43 8037.95   64.39 8082.97   60.06 8127.36   59.98
#Mann= 3 , 0 , 0
       0     .15       0 4394.88    .017       0 4462.39     .15       0
#XS Ineff= 2 , 0
       0    4370            4505       0
Permanent Ineff=
       T       T
Bank Sta=4394.88,4462.39
XS Rating Curve= 0
Exp/Cntr=.3,.1

Type RM Length L Ch R = 1 ,17698   ,624.09,628.37,632.66
BEGIN DESCRIPTION:
17697.70  Survey
END DESCRIPTION:
XS GIS Cut Line= 6
     3072262.459    13799620.585     3074296.887    13797657.709
     3074338.417    13796866.289      3074313.54    13796064.843
     3074322.177    13795977.675      3074190.81     13792269.27
#Sta/Elev= 30
       0   66.84 1167.29    64.3  1313.2   67.13 1624.69   63.64 2021.88   66.17
 2668.02   61.75 2951.44   65.18 3308.24   65.25 3417.99   62.15  3493.1   65.33
  3688.3   62.21  3883.4   65.03 4442.82    61.9 4466.04   50.41 4466.82   46.34
 4474.08   46.34 4474.86   50.34 4509.21   62.67 5669.81   64.63 5816.52   60.72
 5939.98    65.3 6495.33    65.3 6641.23   61.82 6840.54   64.86 6900.58   61.44
 7035.67   65.53 7932.76   65.62  8041.3   61.08 8116.34   63.73 8219.64   57.94
#Mann= 3 , 0 , 0
       0     .15       0 4442.82    .017       0 4509.21     .15       0
#XS Ineff= 2 , 0
       0    4390            4534       0
Permanent Ineff=
       T       T
Bank Sta=4442.82,4509.21
XS Rating Curve= 0
Exp/Cntr=.3,.1

Type RM Length L Ch R = 1 ,17069   ,30.07,35.03,35.09
BEGIN DESCRIPTION:
 17069.33
END DESCRIPTION:
XS GIS Cut Line= 6
     3072331.857    13799600.757     3074385.719    13797691.958
     3074937.277    13796309.471     3074942.353     13796087.64
     3074948.963    13796007.026     3074996.432    13792188.058
#Sta/Elev= 30
       0   67.29  499.17   67.94    1011   63.81 1133.98   66.95 1435.61   64.08
 1669.11    66.1 1789.27   63.05 1870.33   65.73 2075.96   62.85 2399.15    65.1
 2526.47    61.3 2862.53   65.11 3088.63   62.51 3174.27   65.99 3443.92   62.69
 4525.43   62.75 4550.59   50.02 4551.35   45.98 4558.66   45.98 4559.42   50.09
 4594.99   63.81 5739.06    63.8 5916.86   60.15  6124.3   64.45 7072.59   66.32
  7749.9   63.86 8139.41   68.67  8302.4   68.17 8346.85   62.37 8414.39   69.21
#Mann= 3 , 0 , 0
       0     .15       0 4525.43    .017       0 4594.99     .15       0
#XS Ineff= 2 , 0
       0    4470            4609       0
Permanent Ineff=
       T       T
Bank Sta=4525.43,4594.99
XS Rating Curve= 0
Exp/Cntr=.5,.3

Type RM Length L Ch R = 1 ,17034   ,34.45,38.74,38.71
BEGIN DESCRIPTION:
 17034.31
END DESCRIPTION:
XS GIS Cut Line= 6
     3072332.843    13799648.137     3074401.296    13797702.136
     3074961.677    13796309.474     3074977.315      13796089.6
     3074983.925    13796008.986     3075034.025    13792208.818
#Sta/Elev= 30
       0   68.44  994.95   63.85 1159.71    67.1 1393.86   64.01 1680.37   66.09
 1756.96   63.07 1880.53   65.51 2094.22   62.81  2452.7   64.97 2601.35   61.43
 2752.13   64.68    3136    62.3 3251.83   65.94 3491.72   62.72 4574.43   62.75
 4599.59   50.02 4600.35   45.98 4607.66   45.98 4608.42   50.09  4642.4    63.2
 5827.01   63.86 5969.06   60.58 6059.07   64.01 6344.09   65.09 7796.22   64.56
 7979.23   69.05 8092.34   65.71 8339.27   67.91 8373.66    61.6 8442.96   69.23
#Mann= 3 , 0 , 0
       0     .15       0 4574.43    .017       0  4642.4     .15       0
#XS Ineff= 2 , 0
       0    4550            4657       0
Permanent Ineff=
       T       T
Bank Sta=4574.43,4642.4
XS Rating Curve= 0
Exp/Cntr=.5,.3

Type RM Length L Ch R = 3 ,17013   ,,,
BEGIN DESCRIPTION:
Riva Ridge Bridge
END DESCRIPTION:
Bridge Culvert--1,0,-1,-1, 0
Deck Dist Width WeirC Skew NumUp NumDn MinLoCord MaxHiCord MaxSubmerge Is_Ogee
5,32,2.6,0, 8, 8, , , .95, 0, 0,0,,
 4570.64 4582.64 4582.64  4606.9 4631.15 4631.15 4640.06  4642.5
   62.97   62.97   62.97   63.06   62.99   62.99   63.02    63.2
     -.2     -.2   60.84   60.93   60.86     -.2     -.2       0
 4567.64 4579.64 4579.64  4603.9 4628.15 4628.15 4637.06  4639.5
   62.97   62.97   62.97   63.06   62.99   62.99   63.02    63.2
     -.2     -.2   60.84   60.93   60.86     -.2     -.2       0
BR Coef=-1 , 0 , 0 ,, 0 ,,,.8,-1,,0,
WSPro=,,,, 1 ,,,, 0 ,,,, 0 ,,,,-1 ,-1 ,-1 , 0 , 0 , 0 , 0 , 0
BC Design=,, 0 ,, 0 ,,,,,,

Type RM Length L Ch R = 1 ,16996   ,35.92,38.31,38.29
BEGIN DESCRIPTION:
16995.56  Survey
END DESCRIPTION:
XS GIS Cut Line= 6
     3072371.513    13799650.328     3074433.638    13797717.086
     3074990.183    13796319.377     3075015.986     13796091.79
     3075022.596    13796011.177     3075071.299    13792236.774
#Sta/Elev= 30
       0   67.28  662.09   67.66 1043.11   63.78 1113.43   67.13 1248.72   63.47
 1527.31    66.2 1728.94   62.75 1813.83   65.39 2036.69   62.54 2306.96   64.85
 2588.52   61.06 2673.42   64.57  3039.8   62.01 3295.02   65.92 3525.81   62.66
 3652.99   65.07 4571.43   62.75 4596.59   50.02 4597.35   45.98 4604.66   45.98
 4605.42   50.09  4639.4    63.2 5804.65    64.2 5967.56   60.85 6337.82   65.01
 7769.93   64.39 8009.95   69.47 8322.38   66.98    8352   60.73 8415.71   68.38
#Mann= 3 , 0 , 0
       0     .15       0 4571.43    .017       0  4639.4     .15       0
#XS Ineff= 2 , 0
       0    4549            4656       0
Permanent Ineff=
       T       T
Bank Sta=4571.43,4639.4
XS Rating Curve= 0
Exp/Cntr=.5,.3

Type RM Length L Ch R = 1 ,16957   ,143.51,250.54,361.25
BEGIN DESCRIPTION:
 16957.25
END DESCRIPTION:
XS GIS Cut Line= 6
     3072409.736    13799652.717     3074461.504    13797726.251
     3075023.213    13796319.841     3075054.208     13796094.18
     3075060.818    13796013.566     3075109.522    13792239.164
#Sta/Elev= 30
       0   66.91  641.64   67.97   854.6   64.26  970.85    66.9 1013.77   63.84
 1119.89   66.89 1204.79   63.21 1382.36   65.98 1586.81   63.01 2308.27   64.98
 2584.33   61.31 2690.45   64.29 2990.76   61.39 3265.34   65.75 4569.43   62.75
 4594.59   50.02 4595.35   45.98 4602.62   45.98 4603.42   50.09 4639.43   63.83
 5884.29   64.01 6013.71    60.8 6043.71   63.62 6208.72   64.61 7661.51   63.94
 7987.33   68.72  8263.9   65.37 8313.16   67.21  8338.9   60.87 8412.25   69.41
#Mann= 3 , 0 , 0
       0     .15       0 4569.43    .017       0 4639.43     .15       0
#XS Ineff= 2 , 0
       0    4525            4670       0
Permanent Ineff=
       T       T
Bank Sta=4569.43,4639.43
XS Rating Curve= 0
Exp/Cntr=.3,.1

Type RM Length L Ch R = 1 ,16707   ,128.93,222.21,292.49
BEGIN DESCRIPTION:
 16706.75
END DESCRIPTION:
XS GIS Cut Line= 6
     3072440.912    13799660.242     3074482.196     13797752.42
     3075050.698      13796315.4     3075243.635    13796154.502
     3075833.737    13795599.364     3077331.277    13793422.894
#Sta/Elev= 30
       0   66.63  668.12   67.97  787.53   64.41 1018.34   63.98 1103.24   66.97
 1204.92   63.62 1446.56   66.04 1665.22   62.92 1726.82   65.67 1907.88   62.48
 2096.38   65.19 2383.82   61.79 2726.98   64.13 3030.54   61.65 3224.11   65.59
 4175.85   61.25 4628.43   62.75 4653.59   50.02 4654.35   45.98 4661.66   45.98
 4662.42   50.09  4696.4    63.2 4976.88   65.54 5530.56   61.72 5617.02   64.71
    6219   65.18 6469.13   61.95 7547.75   67.12 7806.53   63.86 8042.75   67.99
#Mann= 3 , 0 , 0
       0     .15       0 4628.43    .017       0  4696.4      .1       0
#XS Ineff= 2 , 0
       0    4605            4729       0
Permanent Ineff=
       T       T
Bank Sta=4628.43,4696.4
XS Rating Curve= 0
Exp/Cntr=.5,.3

Type RM Length L Ch R = 1 ,16495   ,22.43,22.85,47.79
BEGIN DESCRIPTION:
 16494.57
END DESCRIPTION:
XS GIS Cut Line= 6
     3072450.116    13799689.855     3074496.929    13797775.604
     3075069.111    13796340.123     3075461.328    13796292.998
     3075900.306    13795950.878     3077449.011    13793489.119
#Sta/Elev= 30
       0   66.92  646.78   67.81  767.46   64.41 1006.29   67.12 1050.21   63.93
 1116.09   67.11 1287.47   64.14 1499.72   65.76 1531.56   62.86 1743.81   65.58
 1899.58   62.31 2060.37   65.03 2380.56   62.12 2550.36   64.31 2631.33   61.66
 2719.17   64.02 2918.84   61.94  3590.4   65.14 4580.93   61.41 4606.34   57.99
 4636.34   48.08 4666.34   46.39 4726.34   64.42  5471.1   63.99 5552.32   61.65
 5889.54    65.1 6498.33   65.13 6780.03    62.1 6853.38   64.55 8210.11   66.54
#Mann= 3 , 0 , 0
       0     .15       0 4580.93     .04       0 4726.34      .1       0
#XS Ineff= 2 , 0
       0    4548            4779       0
Permanent Ineff=
       T       T
Bank Sta=4580.93,4726.34
XS Rating Curve= 0
Exp/Cntr=.5,.3

Type RM Length L Ch R = 3 ,16480   ,,,
BEGIN DESCRIPTION:
Crosswalk Bridge at Patio Glen
END DESCRIPTION:
Bridge Culvert--1,0,-1,-1, 0
Deck Dist Width WeirC Skew NumUp NumDn MinLoCord MaxHiCord MaxSubmerge Is_Ogee
5,6,2.6,0, 7, 7, , , .95, 0, 0,0,,
 4564.82 4591.22 4591.22 4649.72 4708.22 4708.22    4778
   61.34   65.65   65.65    65.7   65.74   65.74   65.27
       0       0   62.35    62.4   62.44       0       0
 4527.82 4554.22 4554.22 4612.72 4671.22 4671.22    4741
   61.34   65.65   65.65    65.7   65.74   65.74   65.27
       0       0   62.35    62.4   62.44       0       0
BR Coef=-1 , 0 , 0 ,, 0 ,,,.8,-1,,0,
WSPro=,,,, 1 ,,,, 0 ,,,, 0 ,,,,-1 ,-1 ,-1 , 0 , 0 , 0 , 0 , 0
BC Design=,, 0 ,, 0 ,,,,,,

Type RM Length L Ch R = 1 ,16472   ,101.14,103.96,107.1
BEGIN DESCRIPTION:
 16471.72
END DESCRIPTION:
XS GIS Cut Line= 6
     3072482.024    13799697.832     3074515.148    13797794.857
     3075093.049    13796355.616     3075461.971    13796315.849
     3076035.437    13796163.131     3077485.803    13793496.477
#Sta/Elev= 30
       0   67.35  697.45   64.68  767.68   67.18   994.6    67.1 1068.89   64.06
 1127.28   67.06 1280.94   64.08 1493.38    65.9 1588.25   62.52 1684.41   65.56
 1864.82   62.35 2034.61   65.25 2342.37   62.16 2586.46   64.35 2641.88   61.54
 3549.57   65.17 4536.82   61.59 4569.29   57.93  4599.3   47.62  4614.3   46.45
 4642.28   50.09  4689.3   64.29 5337.39   64.54 5502.15   61.83 6321.63   65.15
 6852.58   64.36 6941.06   62.04 7226.74   65.65 8182.94   64.79 8337.78   66.86
#Mann= 3 , 0 , 0
       0     .15       0 4536.82     .04       0  4689.3      .1       0
#XS Ineff= 2 , 0
       0    4420            4741       0
Permanent Ineff=
       T       T
Bank Sta=4536.82,4689.3
XS Rating Curve= 0
Exp/Cntr=.5,.3

Type RM Length L Ch R = 1 ,16368   ,207.7,215.79,207.82
BEGIN DESCRIPTION:
 16367.72
END DESCRIPTION:
XS GIS Cut Line= 6
     3072509.944    13799705.809     3074531.823    13797811.099
     3075087.746     13796446.13     3075466.641    13796419.831
     3076122.308    13796272.474     3077529.953    13793503.836
#Sta/Elev= 30
       0   67.79  585.95   65.01  715.17   67.54  984.68   67.07 1065.37   64.11
 1171.49   66.87 1291.79   63.95 1479.24   66.02 1572.68   62.44 1642.78   65.61
 1818.27   62.59 1999.24   65.45 2264.55   62.29  2572.3   64.55 2651.86    61.8
 2877.37   64.53 3061.91   62.28 3428.04   65.14 4466.27   61.44 4526.27   46.79
 4556.27   50.01 4586.27   60.94 4631.42   66.13 5427.71   62.86 6875.49   64.71
 6967.18   62.33 7223.76    65.9 7580.74   64.34 7802.21    66.7 8403.37   66.23
#Mann= 3 , 0 , 0
       0     .15       0 4466.27     .04       0 4586.27      .1       0
#XS Ineff= 2 , 0
       0    4420            4657       0
Permanent Ineff=
       T       T
Bank Sta=4466.27,4586.27
XS Rating Curve= 0
Exp/Cntr=.3,.1

Type RM Length L Ch R = 1 ,16152   ,407.69,402.89,386.8
BEGIN DESCRIPTION:
16151.84  Survey
END DESCRIPTION:
XS GIS Cut Line= 6
     3072525.899    13799717.775     3074544.909    13797831.504
     3075045.591    13796624.859     3075464.385    13796635.613
     3076214.922    13796341.743     3077596.178    13793474.402
#Sta/Elev= 30
       0   67.65  604.34   65.18  807.89   67.61 1069.72   64.13 1157.61   67.34
 1306.69   64.23 1662.97   65.55 1794.81   62.69  1979.7   65.48 2717.64   62.15
 3460.29   65.15 3793.42    61.7 4317.17   61.56 4389.29   44.65  4407.5   44.54
  4421.8   44.84 4466.49   63.84 4626.02   65.93 4913.84    62.7 5576.73   64.57
  5812.7   62.19  6037.3   65.18 6203.79   62.42 6531.86   65.14 7069.58   62.48
 7136.18   65.95 7316.56   66.02 7452.52    62.7 7846.55   67.44 8477.14   66.24
#Mann= 3 , 0 , 0
       0     .15       0 4317.17     .04       0 4466.49     .15       0
#XS Ineff= 2 , 0
       0    4250            4511       0
Permanent Ineff=
       T       T
Bank Sta=4317.17,4466.49
XS Rating Curve= 0
Exp/Cntr=.3,.1

Type RM Length L Ch R = 1 ,15749   ,208.91,210.58,190.11
BEGIN DESCRIPTION:
15748.83  Survey
END DESCRIPTION:
XS GIS Cut Line= 6
     3072579.709     13799729.64     3074585.715    13797882.273
      3075008.83    13797055.704     3075473.802    13797037.768
        3076206.    13796493.221     3077640.328    13793511.194
#Sta/Elev= 30
       0   67.13  445.61   65.46  597.96   68.05 1117.68   64.15 1179.71   67.63
 1723.21   62.81 1892.67   65.55 1934.21   63.22 2583.08   62.68 3355.91   64.38
 3601.29   60.95 3879.73   63.57 3939.85   59.58 3968.58   63.72 4023.44   44.75
 4039.51   44.16 4053.43   44.84 4102.51   63.66 4121.17   65.72 5537.34   61.72
 5694.64   64.53  6099.3   62.49 6871.22   65.27 6926.44   62.43 7032.14   65.66
  7242.7   62.67 7375.86   66.31 7509.02   64.21 7751.44   67.41 8342.71   67.25
#Mann= 3 , 0 , 0
       0     .15       0 3968.58     .04       0 4121.17     .15       0
#XS Ineff= 2 , 0
       0    3929            4138       0
Permanent Ineff=
       T       T
Bank Sta=3968.58,4121.17
XS Rating Curve= 0
Exp/Cntr=.3,.1

Type RM Length L Ch R = 1 ,15538   ,859.18,666.3,492.2
BEGIN DESCRIPTION:
15538.25  Survey
END DESCRIPTION:
XS GIS Cut Line= 6
     3072619.365    13799769.296      3074636.72    13797942.134
     3075038.224    13797252.093      3075474.82    13797247.063
     3076269.184    13796677.797     3077691.837    13793547.986
#Sta/Elev= 30
       0   64.61  427.22    64.7  566.33   68.12  789.34   64.13 1001.73    67.6
 1186.94   63.95 1267.22   67.28 1623.27    63.3 1812.58   65.45 1866.12   62.78
 1957.49   64.97  2493.5   61.96 3018.32   64.68 3091.61   62.31 3779.65   62.64
 3871.45   44.64 3890.83   43.99 3906.16    44.8 3947.33   63.13 3997.84   66.61
 4481.59   62.86 5428.73   61.39 5590.06   64.16 5861.93   62.28 6904.09   65.19
 6994.03   62.04 7356.52   66.53  7587.2   64.21 7684.94   66.99 8372.06   65.53
#Mann= 3 , 0 , 0
       0     .15       0 3779.65     .04       0 3947.33     .15       0
#XS Ineff= 2 , 0
       0    3748            4010       0
Permanent Ineff=
       T       T
Bank Sta=3779.65,3947.33
XS Rating Curve= 0
Exp/Cntr=.3,.1

Type RM Length L Ch R = 1 ,14872   ,757.74,753.39,747.96
BEGIN DESCRIPTION:
14871.95  Survey
END DESCRIPTION:
XS GIS Cut Line= 6
     3072688.763    13799818.867     3075826.723     13798100.27
     3076000.135    13797486.578     3076025.171     13797106.42
     3076254.712    13796920.462     3077772.779    13793570.061
#Sta/Elev= 30
       0   67.55  342.64   68.28  442.09    63.6  574.34   67.26  762.46   64.15
 1105.11   66.38 1324.78   62.03 1425.57   65.44 1480.76   62.62 1668.28   61.82
 2453.24   64.21 2792.45   60.48 3135.94   63.53 3541.89   60.61 3653.38   62.89
 3738.62   60.35 3918.36   63.47 4074.24   60.51 4215.48   62.74 4295.14   44.81
 4319.39   44.32 4330.41   44.61  4380.9    63.5 5916.99   61.53 6740.38   65.09
 7261.88   62.63 7464.97    66.1 7646.12   63.88 8303.79   64.97    8571   71.73
#Mann= 3 , 0 , 0
       0     .15       0 4215.48     .04       0  4380.9     .15       0
#XS Ineff= 2 , 0
       0    4170            4421       0
Permanent Ineff=
       T       T
Bank Sta=4215.48,4380.9
XS Rating Curve= 0
Exp/Cntr=.3,.1

Type RM Length L Ch R = 1 ,14119   ,457.83,464.04,480.19
BEGIN DESCRIPTION:
14118.57  Survey
END DESCRIPTION:
XS GIS Cut Line= 6
     3072708.591    13799838.695     3076217.241    13798251.381
     3076715.861    13797816.472     3076752.194     13797518.27
     3076747.839    13796842.664     3078133.338    13793805.528
#Sta/Elev= 30
       0   67.54   99.94   64.46  204.12   68.04  362.81   67.73  476.17    63.3
  959.18   67.46  1222.6   62.73 1337.84   65.62 1387.23   62.09 1482.83   64.65
 1972.44   62.04 2380.52   64.18 3229.63   60.14 3310.03   63.03 3557.15   63.84
 3853.93   60.58  4191.6   63.12  4435.2   60.15 4594.01   62.65 4688.29   60.05
 4738.27   63.27 4813.05   62.65 4890.31   44.92 4912.32   47.16 4927.19   44.98
 4976.46    63.1 5064.09   65.63 6145.23   61.38 6758.37    65.1 8826.91   64.98
#Mann= 3 , 0 , 0
       0     .15       0 4813.05     .04       0 4976.46     .15       0
#XS Ineff= 2 , 0
       0    4770            5030       0
Permanent Ineff=
       T       T
Bank Sta=4813.05,4976.46
XS Rating Curve= 0
Exp/Cntr=.3,.1

Type RM Length L Ch R = 1 ,13655   ,103.89,103.6,102.2
BEGIN DESCRIPTION:
13654.52  Survey
END DESCRIPTION:
XS GIS Cut Line= 5
     3072728.419    13799848.609      3077041.23    13798173.186
     3077215.952    13797537.825     3077215.952    13797341.664
     3078692.573    13794085.146
#Sta/Elev= 30
       0   66.95  108.32   64.11  304.76   68.07  479.19   63.68  815.29   63.97
  948.45   67.21 1173.74   62.83    1301   65.44 1334.66    61.5 1382.93   64.52
 1522.27   61.91 2042.71   64.54 2251.91   61.05 2472.63   63.87 2976.05   59.99
 3537.88   63.65 3941.58   60.33 4070.32   62.86 4134.68   60.11 5285.76   63.06
 5363.78   44.33 5382.61   43.11 5400.65   44.57 5449.67   62.64 5516.45   65.59
 6649.63   62.43 7792.29   67.87  7816.8   64.07 7873.46   63.17 9057.58   65.76
#Mann= 3 , 0 , 0
       0     .15       0 5285.76     .04       0 5449.67     .15       0
#XS Ineff= 2 , 0
       0    5270            5525       0
Permanent Ineff=
       T       T
Bank Sta=5285.76,5449.67
XS Rating Curve= 0
Exp/Cntr=.3,.1

Type RM Length L Ch R = 1 ,13551   ,80.95,92.39,102.39
BEGIN DESCRIPTION:
 13550.92
END DESCRIPTION:
XS GIS Cut Line= 5
     3072728.419    13799888.265     3077153.574    13798201.232
     3077319.434    13797538.671     3077319.434     13797342.51
     3078788.232    13794129.296
#Sta/Elev= 30
       0   67.25   116.1   63.94  170.58   67.71  302.06   67.64  464.56    63.8
  732.08   66.51  865.88   62.41  952.91   67.53 1170.89    62.6 1283.26   65.18
 1508.01   61.31 2149.65   64.58 2335.96   61.08 2498.67   63.76 2998.42   59.79
 3742.25   63.65 3932.02   60.19 4044.51   62.92 4333.35   60.49 5409.74   63.14
 5440.22   61.47 5505.33   43.87 5615.16   63.18 6771.84   62.64  7349.1   64.07
 7496.25   67.34 7913.01   66.47 7994.28   62.56 8352.47      67    9148   66.56
#Mann= 3 , 0 , 0
       0     .15       0 5409.74     .04       0 5615.16     .12       0
#XS Ineff= 2 , 0
       0    5394            5677       0
Permanent Ineff=
       T       T
Bank Sta=5409.74,5615.16
XS Rating Curve= 0
Exp/Cntr=.5,.3

Type RM Length L Ch R = 1 ,13459   ,108.82,111.35,113.99
BEGIN DESCRIPTION:
 13458.52
END DESCRIPTION:
XS GIS Cut Line= 5
     3072748.248    13799927.921     3077172.125    13798239.905
     3077404.367    13797540.749     3077420.881     13797348.17
     3078876.532    13794195.521
#Sta/Elev= 30
       0   67.43  138.34   63.74  281.69   67.62  443.38   63.98  700.26   66.55
   886.8   62.31  979.76   66.76  1149.8   62.92 1230.07   65.45 1723.49   61.43
 2257.58    64.4 2915.83   59.51 3100.77    62.5 3303.91   59.56 3718.58    63.1
 3942.29   60.22 4184.17   63.21 4547.33   60.85  4875.6   63.51 5482.23   62.38
 5496.22   61.47 5561.33   43.87 5657.56   62.14 7312.39   64.05 7516.62   67.41
 7989.78   63.93 8022.83   65.96 8055.87   63.12 8171.52   66.43 9137.47   67.77
#Mann= 3 , 0 , 0
       0     .15       0 5482.23     .04       0 5657.56     .12       0
#XS Ineff= 2 , 0
       0    5442            5694       0
Permanent Ineff=
       T       T
Bank Sta=5482.23,5657.56
XS Rating Curve= 0
Exp/Cntr=.5,.3

Type RM Length L Ch R = 3 ,13400   ,,,
BEGIN DESCRIPTION:
Fondren Bridge
END DESCRIPTION:
Bridge Culvert--1,0,-1,-1, 0
Deck Dist Width WeirC Skew NumUp NumDn MinLoCord MaxHiCord MaxSubmerge Is_Ogee
5,90,2.6,0, 11, 11, , , .95, 0, 0,0,,
 5383.06 5498.09 5498.09 5508.09 5508.09 5572.18 5636.27 5636.27 5646.92 5646.92
  5668.6
   62.38   62.38   65.34   65.34   63.94   63.89   63.92   65.32   65.32   62.38
   62.14
     -.2     -.2     -.2     -.2   59.15    59.1   59.13     -.2     -.2     -.2
     -.2
    5578 5607.09 5607.09 5617.09 5617.09 5681.18 5745.27 5745.27 5755.92 5755.92
 5777.57
      62   62.14   65.34   65.34   63.94   63.89   63.92   65.32   65.32   62.14
   62.14
     -.2     -.2     -.2     -.2   59.15    59.1   59.13     -.2     -.2     -.2
     -.2
Pier Skew, UpSta & Num, DnSta & Num=  ,5550.82, 2 ,5659.82, 2 , 0 , 0 , 0 ,,
       2       2
       0     100
       2       2
       0     100
Pier Skew, UpSta & Num, DnSta & Num=  ,5593.54, 2 ,5702.54, 2 , 0 , 0 , 0 ,,
       2       2
       0     100
       2       2
       0     100
BR Coef=-1 , 1 , 1 ,1.25, 0 ,,,.8,-1,2,0,
WSPro=,,,, 1 ,,,, 0 ,,,, 0 ,,,,-1 ,-1 ,-1 , 0 , 0 , 0 , 0 , 0
BC Design=,, 0 ,, 0 ,,,,,,

Type RM Length L Ch R = 1 ,13347   ,90.67,98.97,106.2
BEGIN DESCRIPTION:
13347.17  Survey
END DESCRIPTION:
XS GIS Cut Line= 5
     3072728.419    13799987.406     3077194.245    13798274.265
     3077515.019    13797552.179     3077531.533      13797359.6
     3078972.191    13794254.388
#Sta/Elev= 30
       0   67.11  215.96   63.31   288.2   66.59   362.7   64.31   552.7   66.56
  655.86   61.98  924.27   62.28 1017.16   66.34 1155.75   62.59 1249.39   65.29
 1316.41    62.4 1377.11   64.46 1504.84   62.11 2280.36   64.41 2922.99   59.43
 3223.34   62.42 3385.91   58.84 3618.14   62.56 5605.22   61.47 5670.33   43.87
 5766.56   62.14 5857.06   64.54  7494.1   64.03 7598.71    66.8 7642.92   64.32
 7655.19   66.38 8105.93   64.61 8122.46   62.02 8216.23   66.36  9189.7   66.64
#Mann= 3 , 0 , 0
       0     .15       0 5605.22     .04       0 5766.56     .12       0
#XS Ineff= 2 , 0
       0    5557            5782       0
Permanent Ineff=
       T       T
Bank Sta=5605.22,5766.56
XS Rating Curve= 0
Exp/Cntr=.5,.3

Type RM Length L Ch R = 1 ,13248   ,78.16,79.4,81.62
BEGIN DESCRIPTION:
 13248.2
END DESCRIPTION:
XS GIS Cut Line= 5
     3072728.419    13800036.976     3077338.458    13798232.617
     3077606.572    13797547.748     3077640.981     13797356.67
     3079067.849    13794283.822
#Sta/Elev= 30
       0   66.58  160.09   66.52  253.58    63.2  589.31   66.42   698.2   61.88
  925.04   62.53 1013.82   66.58 1142.68   62.28 1283.92   64.94 1315.53   61.98
 1376.53   64.44 1480.15    61.9 1619.65   64.07 1974.01   62.17 2509.02   64.08
 2961.73   59.13 3043.43   62.59 3437.21   59.72 3864.94   63.17 3945.48   60.61
 4409.67   63.19 4605.91   60.53 5532.61   63.94 5589.67   61.25  5683.1   64.92
 5713.22   61.47 5778.33   43.87 5874.56   62.14 5898.92   63.52 9268.17   66.44
#Mann= 3 , 0 , 0
       0     .15       0  5683.1     .04       0 5898.92     .12       0
#XS Ineff= 2 , 0
       0    5667            5987       0
Permanent Ineff=
       T       T
Bank Sta=5683.1,5898.92
XS Rating Curve= 0
Exp/Cntr=.3,.1

Type RM Length L Ch R = 1 ,13169   ,490.92,637.43,748.73
BEGIN DESCRIPTION:
13168.80  Survey
END DESCRIPTION:
XS GIS Cut Line= 5
     3072738.333    13800056.804     3077358.921    13798252.743
     3077684.464    13797558.805     3077718.873    13797367.727
     3079141.433    13794313.255
#Sta/Elev= 30
       0   66.66   133.3   66.94  238.16    63.4  423.15   66.09  503.66   62.68
  597.17   66.21   745.2   61.96 1018.95   66.02 1083.36   65.94 1141.49   62.04
 1276.59   64.91  1308.8   61.74 1357.11   64.41 1488.92   61.57 1566.44   63.97
  2468.2   64.17 2913.39   59.77  3047.9   62.45 3476.22   60.03 3863.04   63.06
 5233.83   61.24 5751.04   65.11 5817.42   42.39 5935.14   64.18 8270.87   63.92
 8294.59   66.49 8320.52   64.01 8585.27   68.34 9062.27   65.22 9290.45   67.11
#Mann= 3 , 0 , 0
       0     .15       0 5751.04     .04       0 5935.14     .12       0
#XS Ineff= 2 , 0
       0    5722            5987       0
Permanent Ineff=
       T       T
Bank Sta=5751.04,5935.14
XS Rating Curve= 0
Exp/Cntr=.3,.1

Type RM Length L Ch R = 1 ,12531   ,689.44,750.52,832.12
BEGIN DESCRIPTION:
12531.37  Survey
END DESCRIPTION:
XS GIS Cut Line= 6
     3072748.248    13800106.374     3077450.926    13798247.473
     3078186.201    13797588.951     3078404.246    13797485.668
     3078790.015    13797032.494     3079461.576    13796530.453
#Sta/Elev= 30
       0   66.51  219.63    63.5  441.69    66.5  526.09    62.6  591.96   65.36
  671.25   62.68  913.19   62.82 1009.97   66.18 1135.28   62.15 1248.27   65.52
  1300.3   61.92 1348.69    64.6 1461.59   61.77  1620.8   64.19 2139.02   61.71
 2534.03   63.78 2913.23   59.82 3329.29   62.64 3526.15    59.9 4279.57   63.11
 4751.98   60.81  5881.1   66.46 6098.54   63.88 6172.48   41.98 6239.68   62.48
 6310.91   65.32 6406.68   62.46 6714.34    61.6 6960.57   64.85 7718.68   64.14
#Mann= 3 , 0 , 0
       0     .15       0 6098.54     .04       0 6239.68     .12       0
#XS Ineff= 2 , 0
       0    6030            6376       0
Permanent Ineff=
       T       T
Bank Sta=6098.54,6239.68
XS Rating Curve= 0
Exp/Cntr=.3,.1

Type RM Length L Ch R = 1 ,11781   ,79.04,80.48,80.31
BEGIN DESCRIPTION:
11780.85  Survey
END DESCRIPTION:
XS GIS Cut Line= 5
      3072777.99    13800136.117     3077407.856    13798292.101
      3078244.63    13798256.908     3078436.886    13798257.333
     3080298.627    13798347.574
#Sta/Elev= 30
       0   66.61  152.52   63.74  441.19   66.44  631.36   62.27  720.66   64.69
  891.52   62.66  995.14   65.95 1108.16   61.86 1214.84   65.67 1269.62   62.11
 1350.35   64.52 1479.52   60.82 1653.62   64.18 2173.24   62.01 2415.06   64.08
 2884.22   59.98 4367.16   63.17 4782.85   61.06 5148.37   63.09 5358.56   60.34
 5463.65   64.08 5684.01   64.47 5850.75   62.18 5909.48   41.81 5918.63   41.13
 6018.97   63.57 6119.04   65.31 6664.73   60.84 7113.34   60.72 7877.28   63.13
#Mann= 3 , 0 , 0
       0     .15       0 5850.75     .04       0 6018.97      .1       0
#XS Ineff= 2 , 0
       0    5740            6281       0
Permanent Ineff=
       T       T
Bank Sta=5850.75,6018.97
XS Rating Curve= 0
Exp/Cntr=.5,.3
